--- LAURELRN3.prj (project) ---

Proj Title=LAURELRN3
Current Plan=p01
Default Exp/Contr=0,0
English Units
Geom File=g01
Flow File=f01
Plan File=p01
Background Map Layer=Inundation Boundary (01pct Value_0)
BEGIN DESCRIPTION:
----------MODEL BY WOOD PLC 2021----------
Stream Name: Laurel Run III
Flood Zone: Enhanced Approximate
Pocahontas County, WV
HEC-RAS Version: RAS 6.1
Vertical Datum: NAVD88
Projection: NAD 1983 StatePlane West Virginia S FIPS 4702 (US Feet)
Terrain: 1-meter LIDAR (FEMA Region III 3DEP collected 2016-2018)
Land Use: 2019 NLCD
Hydrologic Method:
WV SIR2010-5033 regression equations
END DESCRIPTION:
DSS File=dss
DSS Export Rating Curves= 0
DSS Export Rating Curve Sorted= 0
DSS Export Volume Flow Curves= 0
DXF OffsetX= 0
DXF OffsetY= 0
DXF ScaleX= 0
DXF ScaleY= 0

--- LAURELRN3.p01 (plan) ---

Plan Title=Floodplain
Program Version=6.10
Short Identifier=Floodplain
Geom File=g01
Flow File=f01
Subcritical Flow
K Sum by GR= 0
Std Step Tol= 0.01
Critical Tol= 0.01
Num of Std Step Trials= 20
Max Error Tol= 0.3
Flow Tol Ratio= 0.001
Split Flow NTrial= 30
Split Flow Tol= 0.02
Split Flow Ratio= 0.02
Log Output Level= 0
Friction Slope Method= 1
Unsteady Friction Slope Method= 2
Unsteady Bridges Friction Slope Method= 1
Parabolic Critical Depth
Global Vel Dist= 0 , 0 , 0
Global Log Level= 0
CheckData=True
Encroach Param=-1 ,0,0, 0
Computation Interval=0.1SEC
Output Interval=1SEC
Instantaneous Interval=Max Profile
Mapping Interval=1HOUR
Computation Time Step Use Courant=        0
Computation Time Step Use Time Series=    0
Computation Time Step Count To Double=0
Computation Time Step Max Doubling=0
Computation Time Step Max Halving=0
Computation Time Step Residence Courant=0
Run HTab= 0
Run UNet= 0
Run Sediment= 0
Run PostProcess= 0
Run WQNet= 0
Run RASMapper=-1
UNET Theta= 0
UNET Theta Warmup= 0
UNET ZTol= 0
UNET ZSATol= 0
UNET MxIter= 0
UNET Max Iter WO Improvement= 0
UNET MaxInSteps= 0
UNET DtIC= 0
UNET DtMin= 0
UNET MaxCRTS= 0
UNET WFStab= 0
UNET SFStab= 0
UNET WFX= 1
UNET SFX= 1
UNET Gravity=32.174
UNET 1D Methodology=Finite Difference
UNET DSS MLevel= 1
UNET Pardiso=0
UNET DZMax Abort= 0
UNET Use Existing IB Tables= 0
UNET Froude Reduction=False
UNET Froude Limit= 0
UNET Froude Power= 0
UNET D1 Cores= 0
UNET WindReference=Eulerian
UNET WindDragFormulation=Hsu (1988)
UNET D2 Coriolis=0
UNET D2 Cores= 0
UNET D2 Theta= 1
UNET D2 Theta Warmup= 1
UNET D2 Z Tol= 0.01
UNET D2 Volume Tol= 0.01
UNET D2 Max Iterations= 20
UNET D2 Equation= 0
UNET D2 RampUpFraction=0.1
UNET D2 TimeSlices= 1
UNET D2 Turbulence Formulation=Non-Conservative (original)
UNET D2 Eddy Viscosity=0.3
UNET D2 Transverse Eddy Viscosity=0.1
UNET D2 Smagorinsky Mixing=0
UNET D2 BCVolumeCheck=0
UNET D2 Cores=0
UNET D2 SolverType=PARDISO (Direct)
UNET D2 Minimum Iterations= 2147483647
UNET D2 Maximum Iterations= 2147483647
UNET D2 Restart Number= 10
UNET D2 Relaxation Coeff=1.3
UNET D2 SOR Precondition Iterations= 10
UNET D2 ILUT Maximum Fill= 8
UNET D2 ILUT Tolerance=1E-08
UNET D1D2 MaxIter= 0
UNET D1D2 ZTol=0.01
UNET D1D2 QTol=0.1
UNET D1D2 MinQTol=1
DSS File=dss
Write IC File= 0
Write IC File at Fixed DateTime=0
Write IC File at Sim End=0
Echo Input=False
Echo Parameters=False
Echo Output=False
Write Detailed= 0
HDF Write Warmup=0
HDF Write Time Slices=0
HDF Flush=0
HDF Compression= 1
HDF Chunk Size= 1
HDF Spatial Parts= 1
HDF Use Max Rows=0
HDF Fixed Rows= 1
Calibration Method= 0
Calibration Iterations= 20
Calibration Max Change=0.05
Calibration Tolerance=0.2
Calibration Maximum=1.5
Calibration Minimum=0.5
Calibration Optimization Method= 1
WQ AD Non Conservative
WQ ULTIMATE=-1
WQ Max Comp Step=1HOUR
WQ Output Interval=15MIN
WQ Output Selected Increments= 0
WQ Output face flow=0
WQ Output face velocity=0
WQ Output face area=0
WQ Output face dispersion=0
WQ Output cell volume=0
WQ Output cell surface area=0
WQ Output cell continuity=0
WQ Output cumulative cell continuity=0
WQ Output face conc=0
WQ Output face dconc_dx=0
WQ Output face courant=0
WQ Output face peclet=0
WQ Output face adv mass=0
WQ Output face disp mass=0
WQ Output cell mass=0
WQ Output cell source sink temp=0
WQ Output nsm pathways=0
WQ Output nsm derived pathways=0
WQ Create Restart=0
WQ Fixed Restart=0
WQ System Summary=0
WQ Write To DSS=0
Sorting and Armoring Iterations= 10
XS Update Threshold= 0.02
Bed Roughness Predictor= 0
Hydraulics Update Threshold= 0.02
Energy Slope Method= 1
Volume Change Method= 1
Sediment Retention Method= 0
Sediment TS Multiplier= 1
Warm Up Method= 0
XS Weighting Method= 0
Number of US Weighted Cross Sections= 1
Number of DS Weighted Cross Sections= 1
Upstream XS Weight=0
Main XS Weight=1
Downstream XS Weight=0
Number of DS XS's Weighted with US Boundary= 1
Upstream Boundary Weight= 1
Weight of XSs Associated with US Boundary= 0
Number of US XS's Weighted with DS Boundary= 1
Downstream Boundary Weight= 0.5
Weight of XSs Associated with DS Boundary= 0.5
Percentile Method= 0
Sediment Output Level= 3
Mass or Volume Output= 0
Output Increment Type= 1
Profile and TS Output Increment= 1
Transport Output Increment 1
XS Output Flag= 0
XS Output Increment= 10
Read HDF5 Sediment Hotstart= 0
Sediment Hotstart Type= 0
Write Gradation File= 0
Read Gradation Hotstart= 0
Write HDF5 File= 1
Write Binary Output= 1
Write DSS Sediment File= 0
DSS Sediment Output Type= 1
SV Curve= 0
Specific Gage Flag= 0
Subcell Erosion Methods= 0
Subcell Deposition Methods= 0
Advection Scheme= 1
Matrix Solver= 0
Implicit Weighting Factor= 1
Maximum Outer Loop Convergence Iterations= 5
Convergence Maximum Absolute= 0.001
Convergence RMSE= 0.0001
Grain Fractions Max Abs Error= 0.001
Max Subgrid Regions= 1
Max Subgrid Length Scale= 3.402823E+38
Initial Layer Thickness= 3.402823E+38
Min Layer Thickness= 3.402823E+38
Max Layer Thickness= 3.402823E+38
Number of Layers= 5

--- LAURELRN3.f01 (steady flow) ---

Flow Title=Flow
Program Version=6.10
Number of Profiles= 6
Profile Names=01pct,10pct,04pct,02pct,0_2pct,01plus
River Rch & RM=LAURELRN3,Main            ,8318
     658     350     464     558     917     973
River Rch & RM=LAURELRN3,Main            ,4709
     737     393     520     625    1020    1090
Boundary for River Rch & Prof#=LAURELRN3,Main            , 1
Up Type= 0
Dn Type= 3
Dn Slope=0.01771
Boundary for River Rch & Prof#=LAURELRN3,Main            , 2
Up Type= 0
Dn Type= 3
Dn Slope=0.01771
Boundary for River Rch & Prof#=LAURELRN3,Main            , 3
Up Type= 0
Dn Type= 3
Dn Slope=0.01771
Boundary for River Rch & Prof#=LAURELRN3,Main            , 4
Up Type= 0
Dn Type= 3
Dn Slope=0.01771
Boundary for River Rch & Prof#=LAURELRN3,Main            , 5
Up Type= 0
Dn Type= 3
Dn Slope=0.01771
Boundary for River Rch & Prof#=LAURELRN3,Main            , 6
Up Type= 0
Dn Type= 3
Dn Slope=0.01771
DSS Import GetInterval= 0
DSS Import GetPeak= 0
DSS Import FillOption= 0

--- LAURELRN3.g01 (geometry) ---

Geom Title=Geometry
Program Version=6.10

River Reach=LAURELRN3       ,Main
Reach XY= 30
 2249547.5404125475728.631839472      2249720.69      475631.294
     2249726.302      475496.512     2249830.667       475419.36
     2249872.205      475158.8352249792.56115418474853.134746139
     2249648.356      474552.487     2249641.549      474273.593
     2249488.676      474100.546     2249522.722      473967.423
     2249475.855      473484.819     2249545.314        473109.9
     2249459.582      473019.621     2249519.507      472887.843
     2249457.324      472489.692     2249533.692      472341.278
     2249459.316      471976.105      2249572.66      471846.089
     2249557.546      471629.031     2249865.606      471073.176
     2249877.665      470976.125 2249776.6694785470728.284117882
2249817.07849798      470615.826     2250066.416      470455.649
     2250261.468      470215.382     2250325.626      470062.566
     2250325.338      469910.361     2250709.014      469158.067
     2250899.511      468920.866     2250891.613      468428.798

Type RM Length L Ch R = 1 ,8318    ,201.6,201.9,206.9
XS GIS Cut Line= 2
2249614.87979942  475769.77133662249397.13183053475625.153817642
#Sta/Elev= 30
       0 2448.46    27.3 2441.99    37.2 2438.89    45.7 2436.97    54.3 2435.18
    58.9  2434.4    71.6 2433.44    84.9 2433.06    89.7 2433.51    94.5 2434.43
   102.3 2435.01   108.9  2435.1   113.7 2435.49   118.5 2435.57   131.2 2436.56
   143.8 2438.07   152.9 2438.72   174.6 2439.52   181.3 2439.27   196.3 2439.68
   201.5 2439.52   204.4 2439.75   210.1 2440.56     213 2441.25   224.6 2445.09
   233.2  2448.7   241.9 2452.05   246.9 2454.27   253.4 2457.48   261.4 2461.79
#Mann= 3 ,-1,0
       0      .1       0    71.6    .045       0    89.7      .1       0
Bank Sta=71.6,89.7
XS Rating Curve= 0 ,0
Exp/Cntr(USF)=0,0
Exp/Cntr=0.3,0.1

Type RM Length L Ch R = 1 ,8116    ,154.1,153.9,154.8
XS GIS Cut Line= 3
2249779.44557275475677.4907744792249648.13863395475592.877158041
2249530.59110819475491.932672731
#Sta/Elev= 30
       0 2468.01    14.2 2462.98    37.2 2453.98      42 2451.66    46.7 2447.57
    56.2 2436.22      67 2427.05      72 2425.8676.684562426.533    83.6 2427.26
    89.5 2426.71     101 2428.19   122.9 2427.03   132.8 2429.46   146.6 2429.89
   156.2 2431.03     168 2430.94   178.7 2429.37   187.8    2430   203.6 2428.99
   229.4 2428.28   247.8 2430.65   252.4 2430.61   258.1 2429.73   266.3 2430.36
   275.1 2434.97   282.7 2440.26     288 2445.43   293.2 2451.45   311.2 2467.57
#Mann= 3 ,-1,0
       0      .1       0      67    .045       076.68456      .1       0
#XS Ineff= 2 , 0
                          137.52         2438.74
Permanent Ineff=
       F       F
Bank Sta=67,76.68456
XS Rating Curve= 0 ,0
Exp/Cntr(USF)=0,0
Exp/Cntr=0.3,0.1

Type RM Length L Ch R = 1 ,7962    ,203.1,196.9,193.3
XS GIS Cut Line= 2
 2249835.9145301475551.2016772652249592.69415731475404.119086961
#Sta/Elev= 30
       0 2455.71       9  2450.8    11.6 2449.06    18.4 2443.69    37.1 2426.77
    42.6  2423.4    46.4 2422.61    47.9 2422.62      58 2423.13    65.7 2424.13
    69.8 2424.28    79.9 2421.85    97.4 2422.92   107.2 2422.64   114.9  2421.4
   119.9 2420.94   126.5  2421.5   135.3    2425     168 2425.62   191.4 2424.27
   202.3 2423.28   205.4 2423.57   212.6  2425.3   216.8 2425.91   242.8 2426.76
     246  2427.4   251.3 2429.86     259 2435.11   265.3 2440.05   284.2 2455.88
#Mann= 3 ,-1,0
       0      .1       0   114.9    .045       0   126.5      .1       0
#XS Ineff= 2 , 0
           51.21 2430.02  142.03         2430.79
Permanent Ineff=
       F       F
Bank Sta=114.9,126.5
XS Rating Curve= 0 ,0
Exp/Cntr(USF)=0,0
Exp/Cntr=0.3,0.1

Type RM Length L Ch R = 1 ,7765    ,100,99.6,98.9
XS GIS Cut Line= 2
2249913.15343227 475357.282731392249633.77867974475317.019899407
#Sta/Elev= 30
       0 2455.25    13.1 2446.93    25.7 2438.39    28.8 2435.92    37.4 2428.35
    45.4    2419    49.5 2414.96    53.5 2413.41    57.5 2413.06    64.5 2412.38
    71.6 2413.04    73.7 2413.41    78.7 2415.14     102 2416.59   112.9 2418.24
   122.2 2418.92   130.3  2419.2   142.2 2418.81   158.6 2419.41   178.8 2420.68
   190.9 2420.71     199 2421.54   207.1 2421.87   231.3 2421.93   235.4 2422.88
   251.6 2427.92   259.6 2431.28   265.5 2434.18   271.8 2437.81   282.3 2445.22
#Mann= 3 ,-1,0
       0      .1       0    57.5    .045       0    71.6      .1       0
Bank Sta=57.5,71.6
XS Rating Curve= 0 ,0
Exp/Cntr(USF)=0,0
Exp/Cntr=0.3,0.1

Type RM Length L Ch R = 1 ,7666    ,141.1,134.7,130.3
XS GIS Cut Line= 3
2249945.19935977475278.4004483222249909.04498003475254.571425311
2249645.28234602475226.633950058
#Sta/Elev= 30
       0 2443.26    13.2 2437.42      24 2430.26    34.8 2424.83    45.4 2418.01
    52.2 2414.72    56.2 2413.81    72.3 2413.33    76.4 2412.44    80.4 2410.02
    84.4 2408.68    88.4  2408.5    96.5 2409.02    99.9 2410.24   104.5 2415.06
   108.5 2415.72   144.7 2414.15   160.8 2414.56     197 2417.48   205.1 2417.47
   221.2  2420.2   233.2 2423.23   249.3 2423.25   257.4 2424.11   265.4 2425.73
   273.5 2428.45   281.8 2432.67   289.5 2437.59   301.6  2443.6   308.5 2448.12
#Mann= 3 ,-1,0
       0      .1       0    80.4    .045       0    99.9      .1       0
Bank Sta=80.4,99.9
XS Rating Curve= 0 ,0
Exp/Cntr(USF)=0,0
Exp/Cntr=0.3,0.1

Type RM Length L Ch R = 1 ,7531    ,140.5,139.9,139.6
XS GIS Cut Line= 2
2249928.28289471475102.4197710272249648.56910781475163.363785514
#Sta/Elev= 30
       0 2451.73     8.3 2443.91    15.9  2437.3    20.6  2431.9    24.7 2425.49
    28.8 2415.11    29.3 2414.22    31.8 2411.64    32.9 2410.68      37 2408.43
      41 2407.27    49.2 2405.83    57.4 2404.73    69.7 2405.01    73.8 2405.46
   120.1 2409.84   131.1 2411.32   155.7 2411.47   159.8 2412.13   173.8 2415.69
   180.2 2416.79   204.8 2418.64   217.1  2418.9   229.4 2419.72   237.6 2420.97
   247.8 2424.41   253.9 2427.09   262.1  2431.6   274.7 2439.19   286.3 2446.82
#Mann= 3 ,-1,0
       0      .1       0    49.2    .045       0    73.8      .1       0
Bank Sta=49.2,73.8
XS Rating Curve= 0 ,0
Exp/Cntr(USF)=0,0
Exp/Cntr=0.3,0.1

Type RM Length L Ch R = 1 ,7391    ,118.7,121.6,123.3
XS GIS Cut Line= 3
2249909.74760411474963.5621659912249765.47685519474998.457186991
2249613.34371076475078.218081417
#Sta/Elev= 30
       0 2462.21    30.4 2443.61    34.5 2440.48    38.7 2436.66      51 2424.02
    63.3 2413.73    79.8 2403.23    86.8 2400.29    92.2 2399.16    96.3 2398.98
   108.6 2399.21   110.72399.835   112.7 2400.43   116.8 2402.54   125.1 2403.82
   141.5 2402.13   149.9 2402.16   163.3 2402.92   172.5 2405.51   178.1 2406.56
   195.1 2406.91   204.1 2407.66   216.6 2410.07   235.7 2414.78   246.2 2415.76
   266.3 2418.62   276.4 2422.69   303.5  2437.4   312.5 2441.73   320.2 2446.45
#Mann= 3 ,-1,0
       0      .1       0    86.8    .045       0   110.7      .1       0
#XS Ineff= 2 , 0
                          123.99         2412.14
Permanent Ineff=
       F       F
Bank Sta=86.8,110.7
XS Rating Curve= 0 ,0
Exp/Cntr(USF)=0,0
Exp/Cntr=0.3,0.1

Type RM Length L Ch R = 1 ,7269    ,257.7,257.5,254.4
XS GIS Cut Line= 3
2249907.36344356474858.0190084482249745.10075689474872.687476804
2249665.48693492475009.352878698
#Sta/Elev= 30
       0 2454.98    15.3 2447.52    35.3 2438.57    39.3 2436.52    46.4 2431.89
    51.4 2427.77    55.4 2423.95    63.4  2413.9    67.5 2409.16    75.5  2401.9
    79.5 2398.78    83.5 2397.79    87.5  2397.8    95.6 2398.55   101.6 2398.06
   107.6 2397.39   111.6 2397.34   119.7 2397.93   134.8 2397.99   139.8  2397.5
   147.8 2398.05   159.8 2399.72   166.9 2399.27   175.7 2399.87     182 2399.84
   205.2 2401.88   228.3 2403.19   274.6 2408.68   307.8 2412.96   321.1 2415.15
#Mann= 3 ,-1,0
       0      .1       0   101.6    .045       0   119.7      .1       0
#XS Ineff= 2 , 0
                           159.5         2408.27
Permanent Ineff=
       F       F
Bank Sta=101.6,119.7
XS Rating Curve= 0 ,0
Exp/Cntr(USF)=0,0
Exp/Cntr=0.3,0.1

Type RM Length L Ch R = 1 ,7012    ,182.7,183.9,184.9
XS GIS Cut Line= 2
2249805.94140313474622.275002664 2249524.9232697474695.405452592
#Sta/Elev= 30
       0 2434.45    10.4 2427.78    26.6  2418.1    34.9 2411.38      39 2410.22
    43.2 2408.26    55.6 2397.03    59.7 2394.39    63.8 2392.31      68 2391.76
    84.5 2392.47    92.8 2392.06    96.9 2391.73   105.2 2388.23   122.7 2388.24
     130 2387.39   138.2 2388.19   146.5 2388.23   150.6 2388.81   154.8 2391.25
   187.8 2391.71   204.4 2390.96   212.6 2391.77     225 2392.03   233.3 2395.16
   246.5 2402.37   258.1 2406.03   274.6 2413.96   282.9 2417.24   290.4 2421.15
#Mann= 3 ,-1,0
       0      .1       0   122.7    .045       0   138.2      .1       0
Bank Sta=122.7,138.2
XS Rating Curve= 0 ,0
Exp/Cntr(USF)=0,0
Exp/Cntr=0.3,0.1

Type RM Length L Ch R = 1 ,6828    ,201.5,200.5,202
XS GIS Cut Line= 2
2249751.28041389474455.8883092472249460.40199508474509.298188407
#Sta/Elev= 30
       0 2429.65     7.2 2426.16    27.2 2418.35    31.3 2417.24    39.8 2413.71
    43.8 2411.19    47.9 2407.86    55.3 2400.81      67 2390.96    72.3 2386.84
    76.4 2384.77    92.6 2383.64   104.8  2383.7   121.1 2382.79   125.62383.972
   129.2 2385.95   133.3 2386.49   157.7 2385.78   186.2 2386.22   194.3 2385.55
   203.1 2385.42   222.8 2388.14     239 2389.43   246.4 2390.67   251.2 2391.96
   255.3    2394   263.4 2399.31   267.5 2401.16   275.6 2406.69   295.7 2418.26
#Mann= 3 ,-1,0
       0      .1       0   104.8    .045       0   125.6      .1       0
#XS Ineff= 2 , 0
                          137.04          2391.1
Permanent Ineff=
       F       F
Bank Sta=104.8,125.6
XS Rating Curve= 0 ,0
Exp/Cntr(USF)=0,0
Exp/Cntr=0.3,0.1

Type RM Length L Ch R = 1 ,6628    ,159.2,150.3,149.9
XS GIS Cut Line= 2
2249729.09477178474260.325982474 2249420.1391631474326.061218364
#Sta/Elev= 30
       0 2439.29     9.1  2431.6    45.9  2402.5    54.1 2395.29    62.2 2389.56
    70.5 2381.54    75.7 2378.36    78.6 2377.32    85.8 2376.63    92.5 2377.86
    95.9 2378.66   111.4 2379.53   131.8 2378.35   135.9 2378.58   143.1 2380.14
   148.2 2380.62   156.3 2380.26   164.5 2378.05   172.7 2377.44     185 2378.56
   193.7 2379.97   205.4 2379.79   220.7 2377.89   233.9  2378.9   250.4 2382.31
   258.6 2384.99   287.2 2396.47   291.3 2398.35   299.5 2403.05   315.9 2413.58
#Mann= 3 ,-1,0
       0      .1       0    75.7    .045       0    92.5      .1       0
#XS Ineff= 2 , 0
                          152.33         2392.37
Permanent Ineff=
       F       F
Bank Sta=75.7,92.5
XS Rating Curve= 0 ,0
Exp/Cntr(USF)=0,0
Exp/Cntr=0.3,0.1

Type RM Length L Ch R = 1 ,6477    ,96.2,98.5,103
XS GIS Cut Line= 4
2249685.47365114474101.9731123942249607.09126101474108.896979384
 2249572.7586563474157.9518809222249410.27887771474258.682601576
#Sta/Elev= 30
       0 2431.97    13.4 2423.66    37.4  2409.8    46.4 2402.78    57.5 2392.81
    65.6 2386.59    69.6 2383.85    77.6 2379.69    83.9 2374.76    90.7 2373.23
    97.7 2372.87     123 2374.04   132.7  2375.7     144 2375.93   153.4 2375.02
   161.7 2373.24   175.1 2374.32   182.6 2372.51   195.7 2371.68   199.4 2372.48
   205.2 2374.31   219.3 2375.29   238.1 2375.37   248.8  2376.9   266.3 2382.62
   288.9  2393.2   296.5 2395.35   308.7 2397.21   321.5 2402.84   329.7 2405.62
#Mann= 3 ,-1,0
       0      .1       0   182.6    .045       0   199.4      .1       0
#XS Ineff= 2 , 0
           87.79 2384.68  218.68         2385.08
Permanent Ineff=
       F       F
Bank Sta=182.6,199.4
XS Rating Curve= 0 ,0
Exp/Cntr(USF)=0,0
Exp/Cntr=0.3,0.1

Type RM Length L Ch R = 1 ,6379    ,161.1,159.3,163.7
XS GIS Cut Line= 3
2249677.38191963474072.1740436162249562.92191919 474075.04223957
2249381.43414322474127.106809977
#Sta/Elev= 30
       0 2429.36     9.2 2424.01      49 2402.36    64.6 2393.49    69.2 2390.52
    81.2 2384.78    97.2 2375.61   101.2 2373.83   105.2 2372.78   121.7 2371.96
     134 2372.21   144.3 2371.57   167.3 2372.39   175.6 2370.68   188.1 2370.34
   199.3  2369.9204.61732370.576   208.9 2371.65   213.1 2372.18   221.9 2371.53
   225.2 2371.97   228.4 2373.16   233.9 2376.27   238.1 2379.19   241.3  2382.1
   246.4 2385.96   250.5  2388.5   275.5  2400.1   280.1  2402.8   303.3 2418.27
#Mann= 3 ,-1,0
       0      .1       0   188.1    .045       0204.6173      .1       0
#XS Ineff= 2 , 0
                          215.52         2375.83
Permanent Ineff=
       F       F
Bank Sta=188.1,204.6173
XS Rating Curve= 0 ,0
Exp/Cntr(USF)=0,0
Exp/Cntr=0.3,0.1

Type RM Length L Ch R = 1 ,6219    ,165.3,165.9,166.6
XS GIS Cut Line= 2
2249639.16531713473925.3866958262249371.65942663473963.732250095
#Sta/Elev= 30
       0 2418.01     8.5 2412.92    19.2 2405.87    51.5 2381.73    63.6 2373.22
    71.7 2369.85    75.8 2369.11    91.9 2367.88     104 2367.79  110.032365.692
   112.1 2365.06   120.2 2364.83   128.3  2365.8   135.8  2367.3   140.3  2367.7
   152.5 2366.95   160.6 2367.77   168.6 2367.36   176.8 2366.05   184.9  2366.5
   192.9 2365.19     197 2365.06     201 2365.52   213.1 2367.97   221.2 2372.31
   225.3 2375.18   245.5  2392.5   249.5 2395.35   253.6  2397.5   270.2 2409.42
#Mann= 3 ,-1,0
       0      .1       0  110.03    .045       0   128.3      .1       0
#XS Ineff= 2 , 0
             100 2374.71
Permanent Ineff=
       F       F
Bank Sta=110.03,128.3
XS Rating Curve= 0 ,0
Exp/Cntr(USF)=0,0
Exp/Cntr=0.3,0.1

Type RM Length L Ch R = 1 ,6053    ,141.7,141.4,140.8
XS GIS Cut Line= 3
2249598.99378408473770.1784999742249453.74329998473783.797032363
2249336.50336377473839.007684042
#Sta/Elev= 30
       0 2410.85    14.9 2403.75    63.1  2376.1    78.8 2367.34    83.2 2365.15
    91.2 2363.2697.680812360.641    99.3 2360.06   103.3 2359.47   107.3 2359.41
   115.3 2360.46   123.4 2362.36   139.4 2363.33   156.5 2363.56   160.9 2362.86
   165.3 2361.67   169.1 2361.33   174.1  2361.5     183 2362.49   196.1 2361.49
   200.7  2360.2   202.2 2360.17   218.4 2361.32   222.8 2362.47   226.3 2365.03
   235.3 2372.76   240.5  2377.6   249.3 2386.43   253.3 2389.74   275.5 2405.09
#Mann= 3 ,-1,0
       0      .1       097.68081    .045       0   115.3      .1       0
Bank Sta=97.68081,115.3
XS Rating Curve= 0 ,0
Exp/Cntr(USF)=0,0
Exp/Cntr=0.3,0.1

Type RM Length L Ch R = 1 ,5912    ,109,111.1,113.4
XS GIS Cut Line= 4
 2249583.4729645473626.839166158 2249442.3607899473644.361283835
2249368.94359986473615.9050086252249286.41949262473634.440000298
#Sta/Elev= 30
       0 2411.59    19.4  2402.3    35.6 2395.94    40.9 2393.29    47.7 2388.69
    58.8    2379    79.3 2363.54      88 2358.38    98.3 2354.65   104.1 2353.64
   108.1  2353.6  113.962354.853   124.2 2358.68   136.3 2360.12   140.4 2359.44
   148.8  2356.6   161.7 2355.14     166 2356.06   174.6 2356.53   187.4 2355.33
     196 2355.12   221.7 2359.26     234 2358.21   242.2 2358.03   246.1 2358.52
   256.1 2361.27   262.6 2364.51   270.9 2369.54   287.3 2376.21   305.5 2385.42
#Mann= 3 ,-1,0
       0      .1       0    98.3    .045       0  113.96      .1       0
Bank Sta=98.3,113.96
XS Rating Curve= 0 ,0
Exp/Cntr(USF)=0,0
Exp/Cntr=0.3,0.1

Type RM Length L Ch R = 1 ,5801    ,192.7,193.7,194.9
XS GIS Cut Line= 2
2249594.48772488473533.7842525262249291.73105507473521.737900482
#Sta/Elev= 30
       0 2424.16    18.2 2414.44    54.4  2392.7      76 2380.04    78.4 2378.42
    86.4 2371.46   102.4 2355.58   106.4  2352.9   110.4 2351.47   114.3 2350.82
   118.4 2350.66   130.4 2351.53   138.4 2352.38   146.4 2355.26   150.4 2355.61
   158.4 2355.72   178.5 2355.13   190.5 2353.66   194.5 2353.84   202.5 2355.12
   206.5 2355.21   226.5 2353.58   238.5 2354.52   254.5 2353.82   258.5 2353.93
   262.5 2354.89   278.5 2363.71   290.5 2369.01   298.5 2374.68     303 2376.91
#Mann= 3 ,-1,0
       0      .1       0   110.4    .045       0   130.4      .1       0
#XS Ineff= 2 , 0
                          172.46         2363.17
Permanent Ineff=
       F       F
Bank Sta=110.4,130.4
XS Rating Curve= 0 ,0
Exp/Cntr(USF)=0,0
Exp/Cntr=0.3,0.1

Type RM Length L Ch R = 1 ,5607    ,108.1,109.7,109.3
XS GIS Cut Line= 3
2249580.08916192473376.3031713582249532.28261956473341.017390098
2249285.28215074473312.561114888
#Sta/Elev= 30
       0 2402.61     5.3 2399.57      12 2394.72    24.8 2383.78    32.2 2376.85
    39.4 2372.51    59.4 2354.27    66.6 2349.18    71.6 2347.94    83.7 2348.63
    92.4 2348.11   103.8 2347.27   111.7 2347.98     132 2348.77   148.1 2347.58
   168.2  2347.5   176.3 2348.88   180.3 2348.94   188.4 2348.64   200.5 2346.72
   208.5 2346.95   212.5 2346.47   232.7 2348.16   248.8 2348.37   256.8 2350.98
   268.9 2360.29     277 2365.86     285 2373.95   301.1  2388.4   308.1 2394.05
#Mann= 3 ,-1,0
       0      .1       0    92.4    .045       0   111.7      .1       0
#XS Ineff= 2 , 0
                          211.05         2357.76
Permanent Ineff=
       F       F
Bank Sta=92.4,111.7
XS Rating Curve= 0 ,0
Exp/Cntr(USF)=0,0
Exp/Cntr=0.3,0.1

Type RM Length L Ch R = 1 ,5498    ,82.4,83.3,83.6
XS GIS Cut Line= 2
  2249610.429025473245.0065671642249333.61590625473223.698272873
#Sta/Elev= 30
       0 2390.32    18.3 2381.15    41.8 2369.98    46.4 2367.35    50.4 2364.64
    54.4 2361.31    62.4  2353.1    70.5 2345.31    74.5 2344.24    83.9 2345.15
    98.5 2345.88   110.6 2346.02   122.6 2345.78   130.6 2344.99   134.7 2344.98
   139.8 2346.29   146.7 2346.86   150.7 2346.66   158.7 2344.66   166.7 2344.63
   174.8 2343.66   186.8 2345.04   194.8 2345.47   202.9 2344.55   218.9 2345.42
   230.9 2344.57   234.9 2345.49     239    2348     263 2368.54   277.6 2378.66
#Mann= 3 ,-1,0
       0      .1       0    70.5    .045       0    83.9      .1       0
#XS Ineff= 2 , 0
                          223.75         2354.05
Permanent Ineff=
       F       F
Bank Sta=70.5,83.9
XS Rating Curve= 0 ,0
Exp/Cntr(USF)=0,0
Exp/Cntr=0.3,0.1

Type RM Length L Ch R = 1 ,5414    ,197.6,207,207.8
XS GIS Cut Line= 2
2249619.68450481473167.6038507742249342.79957302473130.967326558
#Sta/Elev= 30
       0 2382.05    12.4 2376.38    35.8 2364.34    39.9 2362.42    64.1 2352.08
    68.1 2349.22    72.1 2344.57    76.2 2341.84    80.1 2341.23    83.7 2341.06
    89.6 2341.45    92.3 2341.57   104.4 2342.99   116.5 2342.65   132.7 2343.14
   144.8 2342.58   148.8 2343.05   160.9 2343.63   185.1 2342.58   193.2 2341.45
   201.2 2340.66   205.3 2340.66   208.4 2341.38   217.4 2344.13   221.4  2345.9
   237.6 2354.23   245.6 2359.34   249.7 2361.35   265.8 2370.17   279.3 2378.14
#Mann= 3 ,-1,0
       0      .1       0    76.2    .045       0    89.6      .1       0
#XS Ineff= 2 , 0
                             200         2352.35
Permanent Ineff=
       F       F
Bank Sta=76.2,89.6
XS Rating Curve= 0 ,0
Exp/Cntr(USF)=0,0
Exp/Cntr=0.3,0.1

Type RM Length L Ch R = 1 ,5207    ,129.2,125.6,119.5
XS GIS Cut Line= 4
2249618.96094834472996.1529324022249502.68809335473016.046727202
 2249442.9299154472989.8669540092249335.47246846472998.669936673
#Sta/Elev= 30
       0 2375.08    23.1  2362.6    39.3 2352.26    46.2 2348.36    51.5 2345.48
    59.6    2342    63.7 2341.06    75.9 2341.11      88 2338.53   120.7 2338.21
   133.8 2336.27   143.3 2336.96   151.3  2335.4     160 2334.83   167.6 2335.44
   181.8 2338.07     190 2337.21     198 2337.89     206 2336.29   214.1 2337.79
   218.1 2337.68   226.1 2337.31   234.1 2335.72   238.1 2335.84   242.2 2337.34
   246.2 2339.57   254.2 2346.03   266.2 2357.14   274.4 2364.02     291 2376.08
#Mann= 3 ,-1,0
       0      .1       0   151.3    .045       0   167.6      .1       0
#XS Ineff= 2 , 0
                          183.09         2345.59
Permanent Ineff=
       F       F
Bank Sta=151.3,167.6
XS Rating Curve= 0 ,0
Exp/Cntr(USF)=0,0
Exp/Cntr=0.3,0.1

Type RM Length L Ch R = 1 ,5082    ,84.4,83.5,82.8
XS GIS Cut Line= 3
 2249632.4487083472890.839116279 2249442.9299154472891.408241783
2249363.82147032472864.090217581
#Sta/Elev= 30
       0 2385.47    20.3 2373.23    40.3 2360.64    60.3 2347.03    68.3 2341.94
    80.3 2333.09    84.3 2331.01    88.3 2330.61    96.3 2331.68   100.3 2331.75
   106.3 2330.88   112.3 2329.58   120.3 2330.59   124.3 2331.67   128.3 2333.55
   132.3 2334.94   136.3 2335.33   144.3 2335.33   152.3 2334.69   172.3 2333.98
   188.3 2334.82   199.7 2332.82   202.9 2332.89   209.4 2334.49   222.1 2336.12
   246.9 2340.62   251.7 2342.18   262.6 2347.84   268.6 2350.61   273.2 2351.88
#Mann= 3 ,-1,0
       0      .1       0   106.3    .045       0   120.3      .1       0
#XS Ineff= 2 , 0
                          160.87          2346.8
Permanent Ineff=
       F       F
Bank Sta=106.3,120.3
XS Rating Curve= 0 ,0
Exp/Cntr(USF)=0,0
Exp/Cntr=0.3,0.1

Type RM Length L Ch R = 1 ,4998    ,127.5,126.6,125.1
XS GIS Cut Line= 2
2249617.65528716472800.3920428242249366.21800988472820.359120725
#Sta/Elev= 30
       0 2378.08     5.5 2374.13    17.5 2364.65    33.6 2351.44    41.6 2344.53
    49.6 2336.83    53.6 2333.58    57.7 2331.56    61.8  2331.1    73.7 2332.08
    77.7 2331.61    81.7 2330.28    93.8 2328.12   105.8 2327.03   109.8 2325.84
   113.8 2325.32   117.9  2325.6   121.52327.444   129.9 2330.95   137.9 2330.37
     150 2331.02     158 2332.37     170 2332.68   186.1  2331.6   198.1 2332.89
   210.3    2335   226.2 2341.08   230.2 2342.16   246.3 2344.78   252.2 2345.21
#Mann= 3 ,-1,0
       0      .1       0   105.8    .045       0   121.5      .1       0
Bank Sta=105.8,121.5
XS Rating Curve= 0 ,0
Exp/Cntr(USF)=0,0
Exp/Cntr=0.3,0.1

Type RM Length L Ch R = 1 ,4872    ,160.7,162.3,163.4
XS GIS Cut Line= 2
2249595.46964505472665.7991473392249355.12518882472707.951867353
#Sta/Elev= 30
       0 2361.98    19.6 2352.19    23.7 2349.57    31.8 2343.28    36.9 2338.79
      44 2331.74      48 2328.74    52.1 2327.64    64.3 2327.41    68.3 2326.31
    72.4 2325.95    80.5 2326.69    96.7 2324.51   104.9 2324.51   121.1 2324.05
     123 2324.82   129.2 2327.45   133.3 2327.82   137.4  2327.8   141.4 2327.15
   145.5 2325.64   149.5 2325.58   153.6  2326.9   157.7 2329.11   161.7 2329.68
   190.2 2328.59   196.9 2329.06   214.5 2334.56   230.8 2341.81     244 2348.68
#Mann= 3 ,-1,0
       0      .1       0   104.9    .045       0     123      .1       0
#XS Ineff= 2 , 0
           82.13 2335.12  133.31            2335
Permanent Ineff=
       F       F
Bank Sta=104.9,123
XS Rating Curve= 0 ,0
Exp/Cntr(USF)=0,0
Exp/Cntr=0.3,0.1

Type RM Length L Ch R = 1 ,4709    ,130.1,141.9,150.6
XS GIS Cut Line= 3
2249600.98708667472571.3584888112249511.43338895472523.971181165
2249325.31258145472534.436938911
#Sta/Elev= 30
       0  2349.4     5.2 2344.53    14.5 2339.58    30.3 2333.61    47.4  2328.8
    64.5 2326.68    81.6 2325.42      88 2324.28   104.6 2322.63   116.9 2322.17
   136.6 2322.47   139.7  2322.2   147.3 2319.16   150.2 2318.44   156.7 2317.72
   160.7 2317.81   164.7 2318.43   171.4  2319.8   180.7 2322.46   184.7  2322.9
   188.7 2322.47   201.1 2323.58   212.8  2323.2   216.8 2323.56   232.8  2323.4
   256.8 2325.37   264.9 2328.11   268.7 2330.05   276.9 2335.41   287.7 2343.44
#Mann= 3 ,-1,0
       0      .1       0   150.2    .045       0   164.7      .1       0
#XS Ineff= 2 , 0
           134.3 2327.12
Permanent Ineff=
       F       F
Bank Sta=150.2,164.7
XS Rating Curve= 0 ,0
Exp/Cntr(USF)=0,0
Exp/Cntr=0.3,0.1

Type RM Length L Ch R = 1 ,4567    ,131.5,116.1,106.3
XS GIS Cut Line= 4
 2249599.5148789472431.9229002652249518.05448196472433.262210905
2249471.38619061472367.8127779222249323.10085227472347.113107571
#Sta/Elev= 30
       0 2357.31     7.3 2352.16    23.3 2337.28    31.3 2327.29    35.3 2323.08
    39.3    2320    43.3 2318.06    55.3  2317.6    67.2  2317.9    85.7 2319.62
    94.3 2317.14    97.2 2316.71   105.8 2315.92   112.3 2316.25   119.2 2315.01
   125.8  2314.5   130.7 2313.89   134.5 2314.48   140.5 2317.27   146.7 2317.86
   165.1 2317.94   189.3 2316.75   197.4 2317.33   229.7 2317.87   245.9 2319.41
   278.2 2320.58   286.3 2321.94     294  2324.3   306.5    2330   311.6 2333.08
#Mann= 3 ,-1,0
       0      .1       0   125.8    .045       0   134.5      .1       0
#XS Ineff= 2 , 0
           84.54 2324.51  200.58         2324.15
Permanent Ineff=
       F       F
Bank Sta=125.8,134.5
XS Rating Curve= 0 ,0
Exp/Cntr(USF)=0,0
Exp/Cntr=0.3,0.1

Type RM Length L Ch R = 1 ,4451    ,188.8,189.4,190.6
XS GIS Cut Line= 2
2249580.67921697472285.685145804 2249330.7209825472327.098344415
#Sta/Elev= 30
       0 2352.68     4.6 2350.19     8.6  2347.2    12.7 2343.66    27.8 2329.02
    32.9 2322.96    41.1 2313.75      45 2311.11    49.2 2310.19    57.3 2310.42
    62.6 2311.04    69.4 2312.61    77.5 2312.46    89.7 2314.26    97.8 2314.09
   105.9 2314.42   118.1 2313.71   122.1 2313.81   134.3 2316.04   142.2 2316.66
   146.5 2316.66   154.6 2316.02   170.8 2316.48   191.1 2318.32   199.2 2318.74
   215.4  2320.5   223.5 2321.71   235.7  2324.4   243.8 2326.63   253.4 2330.29
#Mann= 3 ,-1,0
       0      .1       0      45    .045       0    62.6      .1       0
Bank Sta=45,62.6
XS Rating Curve= 0 ,0
Exp/Cntr(USF)=0,0
Exp/Cntr=0.3,0.1

Type RM Length L Ch R = 1 ,4262    ,172.4,180.2,187.6
XS GIS Cut Line= 4
2249567.08139271472118.8873233842249495.07291821472108.044837734
2249476.85468117472111.4056551432249325.85154883472106.427962871
#Sta/Elev= 30
       0 2337.77       7    2334    15.1 2328.48    19.1 2325.11    31.3 2313.56
    35.3 2310.18    39.3 2308.59    63.3 2308.07    67.7 2307.49      75 2305.57
    79.1 2305.29      88 2305.34      92 2305.64     100 2306.77     112 2307.09
     120 2308.74     124 2309.27   144.1 2308.98   156.1 2309.69   176.1 2309.58
   184.1 2310.54   188.1 2310.51   196.1 2309.34   208.1 2310.24   212.1 2310.94
   216.1 2312.57   220.1 2315.23   228.1  2322.2   240.1 2331.11   242.4 2333.27
#Mann= 3 ,-1,0
       0      .1       0      75    .045       0      92      .1       0
#XS Ineff= 2 , 0
           49.11 2313.99   124.8         2313.87
Permanent Ineff=
       F       F
Bank Sta=75,92
XS Rating Curve= 0 ,0
Exp/Cntr(USF)=0,0
Exp/Cntr=0.3,0.1

Type RM Length L Ch R = 1 ,4082    ,162,150.7,148
XS GIS Cut Line= 3
2249619.92627225472024.2769711922249457.56431767471928.845193193
 2249383.3101807 471879.84366684
#Sta/Elev= 30
       0 2347.18       9  2338.3    31.3 2318.47    50.7 2304.27    55.4 2302.23
      60 2301.84    73.9 2303.28    86.8 2303.87   104.4 2302.87   124.5 2303.52
   134.3 2301.74   142.3 2301.55   148.2 2300.56   152.8  2300.2   162.1  2299.2
   168.6  2300.2   171.6 2301.08     176 2304.21   179.8 2305.83   187.7 2306.45
   199.6 2305.54   216.8 2305.76   226.6 2303.73   233.1  2302.8   242.7 2302.56
   252.6 2301.33   257.1  2301.4   261.9 2302.48   271.5  2307.5   277.3 2310.08
#Mann= 3 ,-1,0
       0      .1       0   152.8    .045       0   168.6      .1       0
#XS Ineff= 2 , 0
           91.79 2311.08  217.39         2313.18
Permanent Ineff=
       F       F
Bank Sta=152.8,168.6
XS Rating Curve= 0 ,0
Exp/Cntr(USF)=0,0
Exp/Cntr=0.3,0.1

Type RM Length L Ch R = 1 ,3931    ,63.5,61.2,60.2
XS GIS Cut Line= 2
2249676.40535898471828.6767029682249392.94193668 471831.72542172
#Sta/Elev= 30
       0  2366.1     8.2 2362.23    12.2 2359.92    16.6 2357.23    28.2 2349.38
    32.2 2346.44    60.1 2323.53    76.6 2308.34    84.2 2300.59    87.8  2297.8
    88.2 2297.49    92.2 2297.07   104.2 2297.45   116.2 2298.69   132.2 2298.23
   152.2 2298.76   157.4 2298.58   160.2 2298.67   168.2 2299.88   182.8 2300.13
   196.2 2300.71   204.2 2300.72   212.2 2301.25   216.2 2301.23   224.2 2300.11
   240.2 2300.41   252.2 2299.81   260.2 2300.72   268.2 2302.57   283.5 2311.21
#Mann= 3 ,-1,0
       0      .1       0    87.8    .045       0   104.2      .1       0
#XS Ineff= 2 , 0
                           171.5         2316.01
Permanent Ineff=
       F       F
Bank Sta=87.8,104.2
XS Rating Curve= 0 ,0
Exp/Cntr(USF)=0,0
Exp/Cntr=0.3,0.1

Type RM Length L Ch R = 1 ,3870    ,126.8,137,140.1
XS GIS Cut Line= 4
2249674.54610326471775.8723342492249598.33645478471765.146453869
2249508.91546618471777.4619193652249390.87861457471765.651618417
#Sta/Elev= 30
       0 2358.19    10.5 2352.29    18.6 2347.15    30.7 2338.19    43.4 2327.35
      67 2305.55    70.1 2302.85    75.1 2299.07    79.1 2297.31    89.6 2293.51
    91.3    2293    99.3 2292.55   107.5 2293.32   119.5 2293.83   127.6  2295.1
   135.6 2295.62   147.8 2295.24   159.9 2296.68   176.7 2296.08   196.1 2297.25
   204.1 2298.29   215.7 2297.83   228.3  2298.4   236.3 2300.11   252.4  2305.1
   256.4 2306.05   263.2 2307.12   268.5 2308.43   280.5 2312.14   285.9 2314.17
#Mann= 3 ,-1,0
       0      .1       0    89.6    .045       0   107.5      .1       0
#XS Ineff= 2 , 0
                          158.94         2306.52
Permanent Ineff=
       F       F
Bank Sta=89.6,107.5
XS Rating Curve= 0 ,0
Exp/Cntr(USF)=0,0
Exp/Cntr=0.3,0.1

Type RM Length L Ch R = 1 ,3733    ,137.5,144.4,146.8
XS GIS Cut Line= 2
2249675.33795665 471671.882380682249428.33780779471595.711676092
#Sta/Elev= 30
       0 2334.77     7.5 2328.74    20.1 2318.09      31  2309.7    49.4 2294.02
    53.5 2291.27    57.7 2289.76    61.9 2289.97    68.7 2290.78    78.7 2290.55
    91.2 2291.37   103.8 2290.29     108 2289.57   119.9 2288.84   124.7 2289.19
   127.8 2289.88   137.3 2292.31   141.4 2293.01     154 2293.56   166.6 2295.26
   170.7 2295.42   177.5 2295.18   183.3  2295.6   204.2 2296.09   208.4 2296.37
   212.8    2297   216.8 2297.72   233.5 2302.37   241.9 2305.78   258.5 2313.12
#Mann= 3 ,-1,0
       0      .1       0     108    .045       0   127.8      .1       0
Bank Sta=108,127.8
XS Rating Curve= 0 ,0
Exp/Cntr(USF)=0,0
Exp/Cntr=0.3,0.1

Type RM Length L Ch R = 1 ,3588    ,169.7,167,164.7
XS GIS Cut Line= 3
2249715.04363393 471570.89758315 2249606.3682801471495.277123016
2249501.60275876471448.262598527
#Sta/Elev= 30
       0 2337.99     8.4 2332.74    20.5 2322.97      31 2315.03    37.6 2309.54
      45 2301.73    52.2 2295.83    60.8 2288.17      62 2287.41    63.6 2287.18
    66.5 2287.07    71.7 2287.83    75.1 2287.54    81.5 2285.2483.388692284.977
     101 2284.59   103.9 2285.14   118.2 2287.55   125.3 2288.25   130.2 2288.48
   143.6 2288.09   153.8 2289.19   165.5 2288.56     183 2290.49   196.2 2290.03
   223.4 2291.64   229.5  2292.9   235.6  2295.8   244.4 2298.48   247.2 2300.09
#Mann= 3 ,-1,0
       0      .1       083.38869    .045       0   103.9      .1       0
#XS Ineff= 2 , 0
                          132.85         2296.99
Permanent Ineff=
       F       F
Bank Sta=83.38869,103.9
XS Rating Curve= 0 ,0
Exp/Cntr(USF)=0,0
Exp/Cntr=0.3,0.1

Type RM Length L Ch R = 1 ,3421    ,196.2,199.9,205.4
XS GIS Cut Line= 2
2249789.96377423471405.6546753252249551.09836082471295.465986164
#Sta/Elev= 30
       0 2321.39    13.8 2310.41    29.8 2298.24    32.8    2296    40.9 2290.75
    46.9 2287.62    59.2 2282.53      62 2281.67      68 2280.97      71 2280.96
    81.3 2281.55    92.1 2282.73    98.9 2283.05   107.7 2282.91   125.3 2282.19
   134.1 2284.06   140.4 2283.69   149.4 2283.78   160.6 2284.68     165  2284.8
   191.4 2283.61   211.2  2283.7   215.7 2283.93   218.8 2284.33   221.8 2285.12
   230.8 2288.61   235.4    2290   253.1 2293.53   257.5 2294.67   263.1 2296.42
#Mann= 3 ,-1,0
       0      .1       0      62    .045       0    81.3      .1       0
#XS Ineff= 2 , 0
                          150.72         2290.49
Permanent Ineff=
       F       F
Bank Sta=62,81.3
XS Rating Curve= 0 ,0
Exp/Cntr(USF)=0,0
Exp/Cntr=0.3,0.1

Type RM Length L Ch R = 1 ,3221    ,125.7,121.1,110.4
XS GIS Cut Line= 3
2249874.79485941471263.0624548362249756.02646694471164.261764914
2249611.20166298471165.431727335
#Sta/Elev= 30
       0 2333.82     8.6 2329.02    20.2 2321.49    40.5 2306.09    45.8 2300.89
    51.5 2294.84    57.2 2288.24    60.6 2283.89    65.8 2278.76    68.5 2277.79
      71  2277.3    76.3 2277.03    82.7 2276.82    96.8 2277.18     103 2277.98
   111.1 2276.73   115.5 2276.31   134.3 2276.77   143.9  2278.1   149.1 2278.31
   162.3 2278.31   182.3  2277.6   206.8 2278.97   214.3 2279.06   230.3 2278.47
   238.3 2279.69   258.4 2281.79   278.3 2284.96   282.5 2285.88   299.3 2291.19
#Mann= 3 ,-1,0
       0      .1       0   111.1    .045       0   134.3      .1       0
#XS Ineff= 2 , 0
                          157.49         2286.89
Permanent Ineff=
       F       F
Bank Sta=111.1,134.3
XS Rating Curve= 0 ,0
Exp/Cntr(USF)=0,0
Exp/Cntr=0.3,0.1

Type RM Length L Ch R = 1 ,3100    ,175.6,171.9,164.5
XS GIS Cut Line= 5
2249933.43092656 471139.426969972249891.27820655471107.627549608
2249793.76340657471089.1660424882249737.16313352471102.828177363
2249626.36485593471095.511727766
#Sta/Elev= 30
       0 2325.19    11.6 2317.44    36.9 2298.23      56 2284.67    72.2 2275.27
    76.3 2273.46   82.872272.442    88.5 2271.46    92.6 2271.38   102.1 2272.62
   108.9 2274.94   129.2 2274.73   137.4  2273.9   145.5 2275.18   153.7 2274.75
     166 2272.34   170.1 2272.07   174.3 2272.32   194.8 2275.72     203 2276.46
   215.3 2276.29   239.3 2278.15   251.4 2277.74   263.4 2278.02   279.4 2276.54
   286.8 2276.71   291.4 2277.57   299.5 2280.73   307.5 2285.35   321.3 2294.45
#Mann= 3 ,-1,0
       0      .1       0   82.87    .045       0   102.1      .1       0
Bank Sta=82.87,102.1
XS Rating Curve= 0 ,0
Exp/Cntr(USF)=0,0
Exp/Cntr=0.3,0.1

Type RM Length L Ch R = 1 ,2928    ,149.4,151.6,152.1
XS GIS Cut Line= 4
2249992.97896431470964.4732024842249902.75430991470925.966353268
2249768.18816429470958.2064702752249664.88517814470941.769184731
#Sta/Elev= 30
       0 2295.06    22.6  2279.6      27 2276.99    31.3  2275.7    70.5 2273.86
   126.1 2272.79   129.5 2272.34   133.7 2269.19   137.8 2267.86     146 2267.12
   152.7 2267.68   158.3 2268.91   166.6 2268.82   174.8 2269.76   191.2 2269.03
   207.7 2271.11   215.9 2270.33   224.1 2271.34   236.5 2271.69   244.4 2271.28
   248.6  2270.3   268.8 2270.38   279.3 2269.78   289.1 2268.38   297.2 2268.98
   305.3 2270.61   317.5  2272.2     322 2275.08   326.8 2278.95   341.1 2291.77
#Mann= 3 ,-1,0
       0      .1       0   137.8    .045       0   152.7      .1       0
Bank Sta=137.8,152.7
XS Rating Curve= 0 ,0
Exp/Cntr(USF)=0,0
Exp/Cntr=0.3,0.1

Type RM Length L Ch R = 1 ,2777    ,83.4,88.7,96.9
XS GIS Cut Line= 4
2250041.40105151470830.3070231972249926.03571253 470777.80100353
2249774.79872012470802.4911553712249682.14410533470783.193307016
#Sta/Elev= 30
       0  2286.1    58.5  2279.3    68.2 2276.86    80.3 2272.35    84.8 2271.61
   102.4 2270.67   128.6 2270.36   155.7  2268.7   185.4 2267.64   197.5 2266.56
   217.8 2266.69   225.9 2265.36   242.1 2264.93     247 2263.47   254.3 2262.57
   262.4 2262.72   265.4 2263.45   270.7 2265.63   278.6 2266.88   282.7 2266.54
   290.8 2263.96   294.9 2263.34   311.3 2262.72   313.8 2264.09   315.4 2265.09
   319.4  2270.1     334 2284.18   352.1 2300.66   360.3 2312.44   374.6 2325.54
#Mann= 3 ,-1,0
       0      .1       0     247    .045       0   265.4      .1       0
Bank Sta=247,265.4
XS Rating Curve= 0 ,0
Exp/Cntr(USF)=0,0
Exp/Cntr=0.3,0.1

Type RM Length L Ch R = 1 ,2688    ,57.6,58.8,60.2
XS GIS Cut Line= 4
2250023.06181652470803.9601677752249840.90427833 470728.30602893
2249805.64798062470723.1644855142249716.03822392470691.580718811
#Sta/Elev= 30
       0 2282.33    19.6 2280.26    28.1 2278.85    34.9 2276.89    50.8 2271.23
    59.4 2271.03    77.8 2269.54      90 2269.98    98.4 2269.87   120.1  2268.5
   128.7 2267.44   141.7 2267.12   154.7 2265.97   180.7  2265.4   206.1 2263.73
   218.3 2263.54   230.3 2264.07   238.6 2263.85   255.6 2260.29   264.1 2259.78
   268.4 2259.82   273.2 2260.56   276.8 2262.75   285.8 2272.64     292 2279.87
   298.1 2287.08   301.4 2291.64   306.5 2297.56     315  2309.8   327.9 2321.78
#Mann= 3 ,-1,0
       0      .1       0   255.6    .045       0   273.2      .1       0
#XS Ineff= 2 , 0
          229.95 2272.38
Permanent Ineff=
       F       F
Bank Sta=255.6,273.2
XS Rating Curve= 0 ,0
Exp/Cntr(USF)=0,0
Exp/Cntr=0.3,0.1

Type RM Length L Ch R = 1 ,2629    ,73.9,74.6,76.2
XS GIS Cut Line= 3
2250030.52689751470793.8451577472249946.34731788 470726.84508416
2249741.91119591470632.357800896
#Sta/Elev= 30
       0 2281.87    23.5 2279.23    39.2 2274.41    50.5 2269.85    59.2 2268.02
    81.9 2267.14   105.3 2267.32   123.2 2266.79   176.1 2263.82   189.3 2264.33
   211.3 2262.82     229  2262.1   242.2 2260.13     251 2260.73   255.4 2260.63
   259.8 2259.87   264.2 2258.81   268.6 2258.53     273 2258.56   276.2  2259.9
   277.4 2260.31   282.3 2263.41   285.3 2265.86   290.7 2272.38   297.3 2281.12
   302.2 2286.68   312.4 2296.72   321.4 2306.55   330.5 2314.78   332.8 2317.17
#Mann= 3 ,-1,0
       0      .1       0   259.8    .045       0   276.2      .1       0
Bank Sta=259.8,276.2
XS Rating Curve= 0 ,0
Exp/Cntr(USF)=0,0
Exp/Cntr=0.3,0.1

Type RM Length L Ch R = 1 ,2555    ,144.8,150.8,161
XS GIS Cut Line= 2
2250060.90807044470732.9839673132249776.64367999470558.297290629
#Sta/Elev= 30
       0 2275.19     5.6 2274.16    17.8  2273.2      29 2271.48    43.1 2267.38
    60.7 2264.64    85.4 2264.05    94.8 2263.05   114.2 2263.14   129.5 2264.14
   132.3 2263.92   141.7 2261.83   144.8 2261.59   188.7 2260.56   207.4 2260.66
   226.2 2257.22   236.5 2258.51   240.3 2258.36   251.7 2256.78     265 2257.13
   273.2 2256.39   277.9 2257.22   279.6 2258.84   287.3 2269.15   289.9 2271.92
   296.6 2277.62   305.2 2283.79   311.5 2290.23   323.2 2300.82   333.6 2309.74
#Mann= 3 ,-1,0
       0      .1       0     265    .045       0   277.9      .1       0
Bank Sta=265,277.9
XS Rating Curve= 0 ,0
Exp/Cntr(USF)=0,0
Exp/Cntr=0.3,0.1

Type RM Length L Ch R = 1 ,2404    ,168.2,158,148.7
XS GIS Cut Line= 4
2250060.10304592470669.4517607812249971.96230163470542.953470371
2249949.33216554470482.7133522422249874.02814131 470409.92623594
#Sta/Elev= 30
       0  2268.5    41.9 2262.41    48.9 2261.95    58.8 2261.86    66.2 2261.14
    78.3 2258.54    83.8 2257.69    89.2 2257.46    97.8 2257.97   117.9 2258.31
   149.6 2257.38   164.6 2257.28   168.9 2256.56   177.1 2252.75     186 2252.18
   194.5 2252.33  197.052252.796   203.1 2254.16   215.9 2255.43   226.1 2255.11
   236.8 2255.41   249.5 2254.84   259.1 2255.94   266.8 2256.16   271.4 2257.17
   282.7  2263.1     294 2272.53   302.5 2279.05   318.6 2293.07   323.3 2296.38
#Mann= 3 ,-1,0
       0      .1       0   177.1    .045       0  197.05      .1       0
#XS Ineff= 2 , 0
                          228.82         2261.98
Permanent Ineff=
       F       F
Bank Sta=177.1,197.05
XS Rating Curve= 0 ,0
Exp/Cntr(USF)=0,0
Exp/Cntr=0.3,0.1

Type RM Length L Ch R = 1 ,2246    ,230.4,231.7,232.7
XS GIS Cut Line= 2
 2250219.0994969470497.2107568982249924.91402763470337.155827262
#Sta/Elev= 30
       0 2299.64    26.1 2284.07    44.3 2274.59    53.4 2270.75    61.2 2268.07
    75.9 2264.02    85.3 2262.15   102.5 2260.11   108.1 2258.79   117.2 2254.02
   130.8 2249.88   137.1 2248.64   144.5 2247.84     149 2247.88   153.6 2248.63
   158.5 2249.65   170.3 2250.26   180.9 2252.48   199.1 2253.88   211.6 2254.29
   220.4  2253.2   232.2 2252.94   241.1 2251.34   244.7 2251.56   258.3 2254.39
   273.5 2254.68   291.2 2256.38   294.8 2257.44   301.4 2261.15   334.9 2286.38
#Mann= 3 ,-1,0
       0      .1       0   137.1    .045       0   153.6      .1       0
#XS Ineff= 2 , 0
                          209.66         2261.19
Permanent Ineff=
       F       F
Bank Sta=137.1,153.6
XS Rating Curve= 0 ,0
Exp/Cntr(USF)=0,0
Exp/Cntr=0.3,0.1

Type RM Length L Ch R = 1 ,2014    ,165.8,164.3,163.5
XS GIS Cut Line= 2
2250290.59332881470287.0045312112250058.05493185 470137.45686956
#Sta/Elev= 30
       0 2283.53    12.4 2275.99    25.6 2267.38    43.6 2255.03    46.5 2252.69
   54.76 2243.15    55.2 2242.62      61 2241.85    69.9 2242.47    74.2 2242.92
    78.3 2243.98    84.1 2246.02    88.5 2246.58      98 2246.61   107.3 2246.13
   114.3  2246.6   124.6 2246.02   143.9 2247.03   150.3 2246.93   158.7 2246.14
   170.9 2245.63   176.7 2245.96   188.2 2247.37   211.5 2246.62   217.3 2246.97
     223 2248.49   231.2    2252   255.2 2263.62   269.4 2270.73   276.5 2274.63
#Mann= 3 ,-1,0
       0      .1       0   54.76    .045       0    69.9      .1       0
#XS Ineff= 2 , 0
                           98.07         2255.38
Permanent Ineff=
       F       F
Bank Sta=54.76,69.9
XS Rating Curve= 0 ,0
Exp/Cntr(USF)=0,0
Exp/Cntr=0.3,0.1

Type RM Length L Ch R = 1 ,1850    ,221.5,218.8,218.4
XS GIS Cut Line= 3
2250397.16838153470151.283277702 2250283.9424509470092.567507797
2250166.27455728470014.052964555
#Sta/Elev= 30
       0 2297.78     5.6 2294.08    23.1 2283.63    28.2 2280.26      32 2277.33
    46.2 2264.83    50.7 2259.88    55.2  2255.7    59.7 2252.11    65.4 2246.68
    68.7 2243.96    73.2 2241.56    82.62239.529   100.2 2239.12   104.8  2239.5
   106.1    2240   109.3 2241.39   113.8 2242.08   132.7 2241.62   148.1 2242.69
   164.4 2241.56   180.2 2241.19   194.6 2241.53   204.2  2241.1     225 2241.07
   233.1 2241.64   237.9 2243.17   241.8 2245.03   261.9 2256.85     269 2260.31
#Mann= 3 ,-1,0
       0      .1       0    82.6    .045       0   106.1      .1       0
#XS Ineff= 2 , 0
                          148.79         2250.44
Permanent Ineff=
       F       F
Bank Sta=82.6,106.1
XS Rating Curve= 0 ,0
Exp/Cntr(USF)=0,0
Exp/Cntr=0.3,0.1

Type RM Length L Ch R = 1 ,1631    ,107.5,107.3,107
XS GIS Cut Line= 2
2250475.99472266469978.2751395252250249.25265798469846.725078679
#Sta/Elev= 30
       0 2281.97    36.8 2262.59    41.4 2259.42    50.4 2252.01    55.3 2249.04
    59.9 2245.15    64.5 2241.66    69.2 2238.77    73.8 2236.67    78.4 2236.31
     109 2235.26   117.7 2236.42   133.9 2236.44   143.2 2235.38   152.4  2235.1
   155.8 2234.31   158.7 2233.09   161.6 2232.12   166.3 2231.41   170.4 2231.64
   173.3 2232.73   175.5 2233.68   180.1 2236.92   184.8 2239.51   198.6  2244.5
   212.5 2250.07   217.4 2252.36   235.6 2262.96   246.5 2268.73   262.1 2278.21
#Mann= 3 ,-1,0
       0      .1       0   158.7    .045       0   173.3      .1       0
#XS Ineff= 2 , 0
          122.22 2248.04
Permanent Ineff=
       F       F
Bank Sta=158.7,173.3
XS Rating Curve= 0 ,0
Exp/Cntr(USF)=0,0
Exp/Cntr=0.3,0.1

Type RM Length L Ch R = 1 ,1524    ,211.5,212.5,213.4
XS GIS Cut Line= 2
 2250508.3412977469869.5857833082250317.70911362469764.409405883
#Sta/Elev= 30
       0 2262.38     4.8 2260.06     9.3 2257.55    27.6 2244.25    36.7 2238.49
    42.2 2235.61    47.5 2233.45    50.4  2232.6    73.3 2233.96    91.9 2233.25
   100.2  2233.3   109.4 2233.67   114.4 2233.58   124.1 2233.02     127 2232.12
  131.582230.216   133.3 2229.66   141.7 2229.37   146.4 2229.59   149.9 2230.43
   150.9 2230.75   160.1 2237.63   162.3  2238.9   169.2 2242.48   173.8 2244.38
   177.1 2246.01   197.7 2257.54   203.6  2261.5   210.3 2266.54   217.7 2271.78
#Mann= 3 ,-1,0
       0      .1       0  131.58    .045       0   149.9      .1       0
#XS Ineff= 2 , 0
           114.2 2242.24
Permanent Ineff=
       F       F
Bank Sta=131.58,149.9
XS Rating Curve= 0 ,0
Exp/Cntr(USF)=0,0
Exp/Cntr=0.3,0.1
